--- HartsRun.prj (project) ---

Proj Title=HartsRun
Current Plan=p01
Geom File=g01
Flow File=f01
Plan File=p01
DSS Export Rating Curves=0
DSS Export Rating Curve Sorted=0
DSS Export Volume Flow Curves=0
DXF OffsetX=0
DXF OffsetY=0
DXF ScaleX=0
DXF ScaleY=0

--- HartsRun.p01 (plan) ---

Plan Title=Floodplain
Program Version=4.00
Geom File=g01
Flow File=f01
K Sum by GR=0
Std Step Tol=0.01
Critical Tol=0.01
Num of Std Step Trials=20
Max Error Tol=0.3
Flow Tol Ratio=0.001
Split Flow NTrial=30
Split Flow Tol=0.02
Split Flow Ratio=0.02
Log Output Level=0
Friction Slope Method=1
Unsteady Friction Slope Method=2
Unsteady Bridges Friction Slope Method=1
Global Log Level=0
CheckData=False
Run HTab=0
Run UNet=0
Run PostProcess=0
UNET Theta=0
UNET Theta Warmup=0
UNET ZTol=0
UNET ZSATol=0
UNET MxIter=0
UNET MaxInSteps=0
UNET DtIC=0
UNET DtMin=0
UNET MaxCRTS=0
UNET WFStab=0
UNET SFStab=0
UNET WFX=0
UNET SFX=0
UNET DSS MLevel=0
UNET DZMax Abort=0
UNET Convert EG Bridges=0
UNET Use Existing IB Tables=0
UNET Froude Limit=0
UNET Froude Power=0
Write IC File=0
Echo Input=False
Echo Output=False
Write Detailed=0

--- HartsRun.f01 (steady flow) ---

Flow Title=NFF Regression Equation
Program Version=4.00
Number of Profiles=1
Profile Names=P100yr
River Rch & RM=HartsRun,Main      ,26935.8
533.5893
River Rch & RM=HartsRun,Main      ,25780.1
584.3071
River Rch & RM=HartsRun,Main      ,22928.8
647.6691
River Rch & RM=HartsRun,Main      ,22529.7
720.9590
River Rch & RM=HartsRun,Main      ,21683
989.2965
River Rch & RM=HartsRun,Main      ,20598.1
1034.766
River Rch & RM=HartsRun,Main      ,18245.9
1114.020
River Rch & RM=HartsRun,Main      ,16027.5
1235.337
River Rch & RM=HartsRun,Main      ,15395.8
1411.972
River Rch & RM=HartsRun,Main      ,12886
1528.262
River Rch & RM=HartsRun,Main      ,11632.5
1640.828
River Rch & RM=HartsRun,Main      ,8552.2
1804.659
River Rch & RM=HartsRun,Main      ,6713.9
1936.648
River Rch & RM=HartsRun,Main      ,1772.1
2143.602
Boundary for River Rch & Prof#=HartsRun,Main      ,1
Up Type=0
Dn Type=3
Dn Slope=0.023755

--- HartsRun.g01 (geometry) ---

Geom Title=USGS 10m DEM
Program Version=4.00

River Reach=HartsRun        ,Main
Reach XY= 30
     2152422.939      259405.069      2152048.68      260728.142
     2152324.162      262335.878     2152236.662      262582.753
     2152755.412      263228.065     2153027.287       263956.19
     2152805.412       264756.19     2152444.475      265051.503
     2152905.115      266584.227      2152578.85      267001.503
      2152553.85      267701.503     2152905.412      268101.503
     2153237.212      269296.421     2153727.287      269859.315
     2153727.287      270114.003     2153489.787      270195.253
     2153646.037       271056.19     2154205.412      271745.253
     2154267.912       272449.94     2154881.975      272842.128
       2155247.6       273987.44       2155472.6      274245.253
     2154905.412      275695.253       2154922.6       277112.44
     2155152.287       277674.94     2154613.615      279055.214
     2154886.532      279430.539     2154349.032      281075.852
     2153028.719      281146.164     2152946.007      281563.907

Type RM Length L Ch R = 1 ,26935.8 ,790.7,793.5,796.2
XS GIS Cut Line= 2
     2152018.213      259459.955     2152816.559      259617.167
#Sta/Elev= 30
       0 2196.83    20.1 2187.06    50.2 2173.43   110.5 2147.82   160.7 2125.76
   190.9 2113.72     231 2099.39   241.1 2096.15   261.2 2091.08   281.3 2084.61
   291.3 2082.34   301.4 2081.17   350.5 2077.84   361.6 2077.32   365.5 2077.37
   411.9 2078.95   462.1 2078.96   532.4 2082.03   542.4 2083.41   552.5  2086.7
   572.6 2095.34   602.7 2105.68   612.8 2109.51   622.8 2113.98   642.9 2124.31
     653 2129.96     663 2136.29   693.1 2158.02   703.2 2164.65   813.7 2229.01
#Mann= 3 , 0 , 0
       0      .1       0   350.5    .045       0   365.5      .1       0
Bank Sta=350.5,365.5
XS Rating Curve= 0 ,0
Exp/Cntr=0.3,0.1

Type RM Length L Ch R = 1 ,26142.3 ,362.6,362.2,361.9
XS GIS Cut Line= 2
     2151915.042      260201.803     2152647.064      260435.166
#Sta/Elev= 30
       0 2271.15    29.9 2262.79    39.9 2258.12    79.8 2233.76    89.8 2226.84
   119.7  2202.9   189.6 2148.49   209.5 2131.31   229.5 2112.49   239.5 2104.53
   249.4 2097.78   269.4 2085.88   289.4 2075.63   299.4 2071.56   329.3 2060.96
   339.3 2058.94   339.5 2058.94   349.2 2059.04   354.5    2060   399.1 2071.15
   409.1 2073.18   429.1 2075.09     479  2077.8   508.9 2081.84   548.8 2089.06
   578.7 2093.57   648.6 2101.42   708.4  2107.4   728.4 2111.34   768.3 2122.13
#Mann= 3 , 0 , 0
       0      .1       0   339.5    .045       0   354.5      .1       0
Bank Sta=339.5,354.5
XS Rating Curve= 0 ,0
Exp/Cntr=0.3,0.1

Type RM Length L Ch R = 1 ,25780.1 ,163.9,157.4,150.8
XS GIS Cut Line= 2
     2151836.435      260548.162     2152499.677      260744.678
#Sta/Elev= 30
       0  2175.8      10 2170.42    30.1 2157.97    70.2 2131.16    90.2 2118.69
   130.3 2095.05   150.4 2084.38   170.4 2075.44   180.4 2071.54   190.5 2068.02
   220.6 2058.94   230.6 2056.26   242.1 2053.98   250.6 2053.17   257.1 2053.15
   260.7 2053.14   270.7  2053.6   310.8 2057.61   350.9 2059.78     381 2062.14
     411 2065.31   461.2 2072.19   471.2 2073.76   481.2 2075.84   531.3 2088.23
   551.4 2092.93   561.4 2094.86   611.5 2103.02   661.7 2109.63   691.7  2114.7
#Mann= 3 , 0 , 0
       0      .1       0   242.1    .045       0   257.1      .1       0
Bank Sta=242.1,257.1
XS Rating Curve= 0 ,0
Exp/Cntr=0.3,0.1

Type RM Length L Ch R = 1 ,25622.7 ,105.8,102.7,99.7
XS GIS Cut Line= 3
     2151658.365      260888.478     2151952.764      260773.027
     2152441.987      260770.141
#Sta/Elev= 30
       0 2121.74    19.8 2116.71    39.5 2110.74    88.9 2094.29   118.6    2085
   148.2 2073.62   158.1 2070.29   177.9  2065.4   187.8 2064.12   197.6 2063.57
   227.3 2063.09   256.9 2061.72   296.5 2058.75   346.2 2055.98   376.1 2053.62
   406.1 2053.07   411.8 2053.09   426.8  2053.8     446  2056.6     456 2056.79
   535.9 2054.39   555.8 2054.55   575.8 2055.79   595.8 2059.02   625.7 2066.05
   655.7 2074.44   705.6 2089.81   725.6 2095.13   745.6 2098.77   805.5 2105.85
#Mann= 3 , 0 , 0
       0      .1       0   411.8    .045       0   426.8      .1       0
Bank Sta=411.8,426.8
XS Rating Curve= 0 ,0
Exp/Cntr=0.3,0.1

Type RM Length L Ch R = 1 ,25520   ,153.4,153.5,153.7
XS GIS Cut Line= 2
     2151664.484      260931.369     2152541.437      260803.633
#Sta/Elev= 30
       0 2115.93    60.4 2101.59   100.7  2091.1   130.9 2082.22   181.3 2065.71
   201.4 2060.71   211.5 2059.11   221.6 2058.24     292 2053.96   352.5 2051.51
   392.8 2048.24   402.8 2047.91   414.2 2048.22   429.2 2048.94   543.8 2052.24
   553.9 2053.04     564 2054.75   584.1  2059.5   604.2 2065.62   614.3 2069.76
   624.4  2074.7   654.6 2090.43   664.7 2094.58   674.7 2097.96   694.9 2103.29
     715 2107.36   735.2 2110.13   795.6 2114.15   825.8 2117.08   886.2 2127.52
#Mann= 3 , 0 , 0
       0      .1       0   414.2    .045       0   429.2      .1       0
Bank Sta=414.2,429.2
XS Rating Curve= 0 ,0
Exp/Cntr=0.3,0.1

Type RM Length L Ch R = 1 ,25366.4 ,212.1,212.7,213.3
XS GIS Cut Line= 2
     2151679.223      261073.843     2152588.109      260960.846
#Sta/Elev= 30
       0 2099.45    40.3 2090.33    90.6 2077.73   120.8 2069.53     151 2059.68
     161 2057.46   181.2 2055.52   291.9 2049.95     436 2045.38     451 2045.22
   493.2 2045.02   503.2  2045.2   513.3 2046.51   523.4  2049.7   533.4 2054.23
   553.6 2064.22   583.8 2080.66   664.3 2128.98   684.4 2140.16   694.5 2144.68
   714.6 2151.29   734.7 2158.95   744.8 2162.02   754.8 2163.84   805.2 2168.92
   815.2 2169.73   875.6 2171.72   885.7 2172.38   895.8 2174.03   915.9 2178.58
#Mann= 3 , 0 , 0
       0     .11       0     436    .045       0     451     .11       0
Bank Sta=436,451
XS Rating Curve= 0 ,0
Exp/Cntr=0.3,0.1

Type RM Length L Ch R = 1 ,25153.8 ,342.9,344.2,345.5
XS GIS Cut Line= 2
     2151637.463      261277.728     2152688.824      261177.014
#Sta/Elev= 30
       0  2080.3    10.1 2077.58    20.1 2076.16    60.4 2074.13    80.5 2072.05
   130.8 2062.28   150.9 2059.12   241.4 2048.86   291.7 2043.79   321.9 2042.45
   491.1 2041.34   506.1 2041.19   563.3 2041.07   573.4 2041.52   583.4 2043.66
   593.5 2048.24   603.5 2054.52   633.7 2077.12   643.8 2083.33   694.1 2111.31
   754.4 2146.92   804.7  2174.3   834.9 2189.43   865.1 2203.65   895.2 2217.04
   905.3  2221.1   915.4  2224.2   935.5 2227.94   945.5 2230.47  1056.2 2266.87
#Mann= 3 , 0 , 0
       0     .11       0   491.1    .045       0   506.1     .11       0
Bank Sta=491.1,506.1
XS Rating Curve= 0 ,0
Exp/Cntr=0.3,0.1

Type RM Length L Ch R = 1 ,24809.6 ,314.1,311.2,308.6
XS GIS Cut Line= 2
     2151511.187      261594.432     2152764.824      261548.921
#Sta/Elev= 30
       0 2113.48    20.1  2107.1    80.3 2093.59   130.5  2084.1   150.5 2079.42
   240.9 2052.66   260.9 2047.26     271 2045.19   301.1 2040.91   331.2 2037.91
   371.3 2035.11   461.6 2031.17   630.7 2031.09   642.3 2031.03   645.7 2031.05
   762.7 2032.34   772.8 2034.16   802.9 2043.51     843 2054.62   933.3 2077.46
   943.4  2079.5   953.4 2080.92   983.5 2082.77  1003.6 2085.98  1033.7  2084.3
  1103.9 2093.82  1154.1 2102.22  1214.3 2113.18  1234.4 2117.45  1254.5 2123.51
#Mann= 3 , 0 , 0
       0     .11       0   630.7    .045       0   645.7     .11       0
Bank Sta=630.7,645.7
XS Rating Curve= 0 ,0
Exp/Cntr=0.3,0.1

Type RM Length L Ch R = 1 ,24498.3 ,396,392.6,388.9
XS GIS Cut Line= 2
     2151718.058       261950.25     2152578.641      261817.853
#Sta/Elev= 30
       0 2064.36      30  2057.8      50 2053.12    70.1 2047.86   120.1  2034.2
   130.1 2031.67   140.1 2029.86   150.1 2028.95   180.2 2028.11   270.2 2026.58
   300.2 2026.76   380.3 2026.47   420.3 2026.86   460.4 2025.84   479.1 2025.12
   494.1 2024.66   500.4 2024.63   510.4 2025.31   550.4 2030.19   560.5 2031.52
   570.5 2033.29   630.5 2045.35   660.5 2051.86   680.6 2056.56   700.6  2061.8
   760.6 2079.38   810.7 2093.46   820.7 2097.15   840.7 2106.12   870.7 2118.34
#Mann= 3 , 0 , 0
       0     .11       0   479.1    .045       0   494.1     .11       0
Bank Sta=479.1,494.1
XS Rating Curve= 0 ,0
Exp/Cntr=0.3,0.1

Type RM Length L Ch R = 1 ,24105.7 ,667,664.3,661.3
XS GIS Cut Line= 2
     2151775.982      262409.504     2152773.099      262090.923
#Sta/Elev= 30
       0 2141.17    40.3 2112.43    60.4 2098.72    80.5 2085.83   100.6 2074.12
   130.8 2059.12     151 2050.56   181.2 2039.35   201.3 2033.75   261.7 2021.47
   271.8 2020.17   442.9 2020.76   483.1 2019.64   520.5 2016.95   535.5 2016.06
   543.5 2015.97   583.8 2018.76   694.5 2035.09   734.8 2041.67     765 2047.49
   785.1  2052.2   815.3 2060.47   835.4 2067.15   845.5 2071.02   865.6 2079.97
   895.8  2096.3     926 2115.42   996.4 2162.66  1026.6 2180.38  1046.8 2190.67
#Mann= 3 , 0 , 0
       0     .11       0   520.5    .045       0   535.5     .11       0
Bank Sta=520.5,535.5
XS Rating Curve= 0 ,0
Exp/Cntr=0.3,0.1

Type RM Length L Ch R = 1 ,23441.4 ,511.4,512.6,514.1
XS GIS Cut Line= 3
     2151925.058      263047.812     2152602.174      262741.602
     2153122.382      262694.316
#Sta/Elev= 30
       0 2182.37    40.2 2161.47    90.4 2140.11   170.7 2103.34   220.9 2080.96
     241 2072.48   271.1 2060.41   311.3 2045.37   351.5 2030.85   361.5 2027.39
   411.7 2011.39   421.8 2009.01   451.6 2004.46     462  2003.9   466.6  2003.9
   522.2 2005.51   642.7 2007.92     703 2009.93   783.3 2013.76   803.4 2015.02
   853.6  2018.6   863.7 2019.82   873.7 2021.54     944 2036.24   974.2 2043.44
  1134.9 2090.78    1155 2097.58  1175.1  2105.2  1215.3  2123.3  1265.5 2144.79
#Mann= 3 , 0 , 0
       0      .1       0   451.6    .045       0   466.6      .1       0
Bank Sta=451.6,466.6
XS Rating Curve= 0 ,0
Exp/Cntr=0.3,0.1

Type RM Length L Ch R = 1 ,22928.8 ,397.4,399.1,400.3
XS GIS Cut Line= 3
       2151799.9      263120.164     2152421.419      263261.812
     2153181.997      262971.639
#Sta/Elev= 30
       0 2201.34    59.8 2174.33   159.4 2133.02   229.1 2102.99   268.9 2084.63
   298.8 2074.74   358.6 2057.58   368.5 2054.15   408.4 2037.76   428.3 2031.37
   448.2 2026.37   468.1  2022.5   478.1 2021.43     508 2021.29   527.9 2020.24
   647.5 2010.96   697.8 2005.83   758.1 1998.52     936 1996.61     949 1996.55
     951 1996.59  1019.4 1999.59  1039.5 2001.68  1059.6 2004.91  1119.9 2016.55
  1270.6 2051.32  1280.7 2054.56  1391.2 2099.97  1421.4 2113.72  1451.5 2128.76
#Mann= 3 , 0 , 0
       0      .1       0     936    .045       0     951      .1       0
Bank Sta=936,951
XS Rating Curve= 0 ,0
Exp/Cntr=0.3,0.1

Type RM Length L Ch R = 1 ,22529.7 ,837.8,846.7,855
XS GIS Cut Line= 4
     2152329.489      264037.204     2152621.882      263582.503
     2152952.571      263483.677     2153398.045      263516.626
#Sta/Elev= 30
       0 2089.27      20 2084.28      40 2079.93   100.1  2067.9   150.2 2056.95
   230.2 2040.13   360.4 2015.91   480.5 1995.43   490.5 1994.49   500.6 1994.35
   570.2 1996.52     580 1996.64   589.9 1996.27   698.4 1986.32   705.3 1986.07
   708.2 1985.96   720.3 1987.04   737.8 1990.31   767.4 1995.08     797 1998.76
   816.7 2000.16     866 2001.84   905.6 2004.86   945.3 2007.32  1004.9 2012.55
  1064.4 2018.99  1153.8 2030.99  1203.4 2038.09  1272.9 2048.95  1332.4 2059.06
#Mann= 3 , 0 , 0
       0      .1       0   705.3    .045       0   720.3      .1       0
Bank Sta=705.3,720.3
XS Rating Curve= 0 ,0
Exp/Cntr=0.3,0.1

Type RM Length L Ch R = 1 ,21683   ,440.6,442.2,444.3
XS GIS Cut Line= 2
     2152321.712      264187.091     2153472.323      264320.991
#Sta/Elev= 30
       0 2102.64    20.2 2093.96    40.3 2084.34   100.7 2052.55   120.9  2042.3
     141  2032.8   161.2 2024.27   191.4 2013.07   221.6  2003.2   302.2 1980.76
   312.3 1979.05   322.3 1978.34   463.4  1974.9   523.8 1972.43   564.1 1970.14
   569.9  1970.2   584.9 1970.67   614.4 1971.93     685 1973.77   725.2 1976.58
   735.3 1977.88   815.9 1993.78   876.3 2003.64   906.6  2008.1   956.9 2014.75
  1027.4 2022.58  1057.6 2025.18  1067.7 2025.48  1097.9 2025.38  1158.4    2026
#Mann= 3 , 0 , 0
       0     .09       0   569.9    .045       0   584.9     .09       0
Bank Sta=569.9,584.9
XS Rating Curve= 0 ,0
Exp/Cntr=0.3,0.1

Type RM Length L Ch R = 1 ,21240.8 ,649.6,642.6,635.5
XS GIS Cut Line= 2
     2152160.761      264503.037     2153360.613      264776.107
#Sta/Elev= 30
       0 2179.11    20.2 2166.21    30.3 2158.92    50.4 2143.42    60.5 2136.08
     121 2094.37   141.2 2081.43   191.6 2050.54   221.9 2033.04   252.2 2017.31
   262.2 2012.58   282.4  2004.1   302.6 1997.05   373.2 1975.27   383.3 1972.66
   393.4 1971.17   413.5 1970.29     464 1969.22   615.3 1967.71   680.9 1964.88
   685.9 1964.76   695.9 1964.92   847.2 1976.32   887.6 1978.64   897.7 1979.55
   917.9 1982.29   978.4 1991.94   998.6 1994.68  1079.2 2002.17  1230.5 2017.31
#Mann= 3 , 0 , 0
       0      .1       0   680.9    .045       0   695.9      .1       0
Bank Sta=680.9,695.9
XS Rating Curve= 0 ,0
Exp/Cntr=0.3,0.1

Type RM Length L Ch R = 1 ,20598.1 ,335.4,331.8,328
XS GIS Cut Line= 2
     2152218.685      265074.001      2153141.33      265057.451
#Sta/Elev= 30
       0 2104.07    20.1 2091.58    30.1 2085.17    50.2 2072.02    90.3 2045.23
   120.4 2024.68   180.6 1983.24   190.6 1975.94   200.6 1967.11   210.6 1958.07
   219.2 1954.05   220.7 1953.35   230.7  1952.7   234.2 1952.79   240.7 1952.96
   260.8  1954.3   300.9  1956.7   310.9 1957.21     331 1957.93   351.1 1958.26
   401.2 1958.42   441.3 1958.99   571.7 1961.68   682.1 1963.38   702.1 1963.78
   712.2 1964.18   722.2 1965.06   732.2 1966.19   862.6 1982.04   922.8 1988.56
#Mann= 3 , 0 , 0
       0     .09       0   219.2    .045       0   234.2     .09       0
Bank Sta=219.2,234.2
XS Rating Curve= 0 ,0
Exp/Cntr=0.3,0.1

Type RM Length L Ch R = 1 ,20266.3 ,553.7,552.2,550.8
XS GIS Cut Line= 2
     2152171.192      265449.215     2152968.926      265303.923
#Sta/Elev= 30
       0 2174.58      30 2156.07    60.1 2135.99    80.1 2121.54    90.1 2113.62
   100.1 2105.16   120.1 2086.53   140.2    2066   180.2 2023.16   200.2 2003.34
   210.2 1994.37   220.2 1986.16   230.2 1978.76   240.2  1972.4   250.3 1967.01
   260.3 1962.53   270.3 1958.82   280.3 1955.85   290.3 1953.54   300.3 1951.92
   310.3 1951.36   330.4 1951.39   357.4 1948.95   370.4 1948.46   372.4 1948.51
   580.6  1954.3   630.7  1955.2   670.7 1955.22   730.8 1959.63   810.9 1967.16
#Mann= 3 , 0 , 0
       0      .1       0   357.4    .045       0   372.4      .1       0
Bank Sta=357.4,372.4
XS Rating Curve= 0 ,0
Exp/Cntr=0.3,0.1

Type RM Length L Ch R = 1 ,19714.1 ,807.3,815.2,820.2
XS GIS Cut Line= 3
     2152093.539      265638.859     2152509.848      265952.047
     2153155.338      265780.918
#Sta/Elev= 30
       0 2163.54    40.1 2136.76    70.1 2114.45    90.2 2100.46   130.2 2075.18
   170.3  2048.6   270.5 1987.24   280.5 1981.65   290.5 1977.23   300.6 1973.94
   320.6 1969.01   350.6 1962.64   360.7  1961.5   410.8 1958.47   470.9 1952.92
   610.7 1943.91   640.6 1939.97   649.3 1939.47   650.5  1939.4   664.3 1939.56
     800 1942.45   869.8 1945.68   899.7  1948.5   939.6 1956.66   959.5 1959.49
   979.4 1961.45  1009.3 1963.29    1099 1967.28  1148.9 1968.75  1188.8 1970.74
#Mann= 3 , 0 , 0
       0      .1       0   649.3    .045       0   664.3      .1       0
Bank Sta=649.3,664.3
XS Rating Curve= 0 ,0
Exp/Cntr=0.3,0.1

Type RM Length L Ch R = 1 ,18898.9 ,652.7,653,653.4
XS GIS Cut Line= 2
      2152289.07      266660.893     2153602.547      266566.309
#Sta/Elev= 30
       0 2061.35    60.3 2027.14   120.6 1994.02   221.2 1941.57   231.2 1937.41
   241.3 1935.19   251.3 1934.45   452.4 1934.11   532.8 1932.97   552.9  1932.3
     583 1930.43   602.8 1927.78   617.8 1926.93   623.3 1926.91   633.3 1927.17
   643.4 1928.27   653.4  1930.6   713.7 1947.84   743.9 1954.99     764 1958.49
   804.2 1963.28   864.5 1966.88     965  1973.8  1055.5 1981.12  1186.2 1981.86
  1206.3 1981.56  1236.5 1980.12  1246.5 1980.37  1286.7 1984.08  1316.9 1990.62
#Mann= 3 , 0 , 0
       0      .1       0   602.8    .045       0   617.8      .1       0
Bank Sta=602.8,617.8
XS Rating Curve= 0 ,0
Exp/Cntr=0.3,0.1

Type RM Length L Ch R = 1 ,18245.9 ,971.1,969.6,967
XS GIS Cut Line= 2
     2152234.177      267147.866     2153328.043      267085.802
#Sta/Elev= 30
       0 2111.51    30.2 2097.49    50.3 2089.23    70.4 2082.14   110.6 2069.58
   130.7 2062.44   150.8  2053.8   170.9 2043.46     191 2031.47     201 2024.91
   211.1 2017.54   221.1 2008.74   241.2 1988.16   251.3 1978.77   261.3 1970.28
   281.4 1954.68   301.6 1940.62   321.6 1925.54   331.7 1920.63   339.4 1919.69
   341.8  1919.4   354.4  1919.6   522.7 1921.43   572.9 1922.36   623.2  1923.7
   743.8 1928.48   814.2 1936.79   874.5 1945.62     975 1954.35  1095.6 1963.88
#Mann= 3 , 0 , 0
       0     .11       0   339.4    .045       0   354.4     .11       0
Bank Sta=339.4,354.4
XS Rating Curve= 0 ,0
Exp/Cntr=0.3,0.1

Type RM Length L Ch R = 1 ,17276.3 ,920.9,918,916.1
XS GIS Cut Line= 2
     2152329.203      268101.924     2153564.537      267801.643
#Sta/Elev= 30
       0 2128.86   161.4 2025.79   171.5 2018.82   181.6 2011.08   191.7 2002.55
   211.9 1984.56     222  1976.1   232.1 1968.52   252.2 1955.03   272.4 1942.27
   292.6  1931.2   312.8 1921.94   322.9 1917.89     333 1914.48     343 1911.98
   353.1 1910.24   373.3 1908.38   460.7 1905.89   464.1 1905.86   475.7 1905.98
   686.1 1909.29   736.6 1910.57   766.8 1912.05   817.3 1916.28   877.8 1919.38
   918.2 1921.96    1130 1929.74  1200.7 1931.56    1241 1933.84  1271.3 1934.45
#Mann= 3 , 0 , 0
       0     .11       0   460.7    .045       0   475.7     .11       0
Bank Sta=460.7,475.7
XS Rating Curve= 0 ,0
Exp/Cntr=0.3,0.1

Type RM Length L Ch R = 1 ,16358.3 ,330,330.8,331.6
XS GIS Cut Line= 2
     2152607.603      268959.037     2153765.991      268637.869
#Sta/Elev= 30
       0 2065.54    50.1 2052.53    70.1 2045.66   110.2 2029.83   130.2 2020.46
   160.3 2003.87   170.3  1998.8   260.4 1957.28   310.5 1935.11   380.7 1906.21
   390.7 1903.47   400.7 1902.15   470.8 1897.62     497 1894.56   510.9 1893.63
     512 1893.66   520.9 1893.89     601 1899.51   721.2 1905.64   791.4 1910.68
   831.4 1915.34   851.5  1918.3   871.5 1922.51   911.6 1931.94   941.6 1937.06
   971.7 1941.14   991.7 1942.61  1031.8 1944.27    1122  1950.5  1202.1 1956.69
#Mann= 3 , 0 , 0
       0     .11       0     497    .045       0     512     .11       0
Bank Sta=497,512
XS Rating Curve= 0 ,0
Exp/Cntr=0.3,0.1

Type RM Length L Ch R = 1 ,16027.5 ,636.3,631.7,627.1
XS GIS Cut Line= 3
     2152656.091      269097.793     2152955.761      269191.479
     2153836.427      268978.134
#Sta/Elev= 30
       0 2062.88    39.2 2049.44    98.1 2023.78   117.7 2012.97   137.4  1999.8
   147.2 1994.24   186.4 1974.31   225.7 1952.78   274.7  1929.5   304.2 1916.64
     314 1913.01     324  1910.3   344.2 1906.15   374.4 1902.26   414.7 1899.64
   553.8 1892.33   565.7    1892   568.8 1892.04   696.6 1898.09     767 1898.89
   797.2 1900.83   817.4 1903.38   837.5  1907.2   867.7 1916.12   887.9 1920.38
   928.1 1927.07   968.4 1932.94  1099.3 1946.25  1159.7 1953.24  1220.1 1958.13
#Mann= 3 , 0 , 0
       0     .11       0   553.8    .045       0   568.8     .11       0
Bank Sta=553.8,568.8
XS Rating Curve= 0 ,0
Exp/Cntr=0.3,0.1

Type RM Length L Ch R = 1 ,15395.8 ,1008.3,1014.7,1020.5
XS GIS Cut Line= 3
     2153078.005      270029.045     2153382.087      269721.162
     2154115.686      269386.671
#Sta/Elev= 30
       0 2027.05    40.2 2004.57   130.8 1958.79   181.1 1934.36   211.3 1920.28
   251.6 1902.14   261.6 1898.19   271.7 1895.98   281.8 1895.18     322 1894.62
   392.5 1894.42   422.7 1893.82   543.6 1889.44   573.8 1887.36   581.3 1887.16
   583.9 1887.09   596.3 1887.84   624.2 1888.55   785.5 1889.33   795.6 1890.68
   815.7 1898.28   825.8  1900.2   906.4 1907.89  1017.3 1916.65  1027.4  1917.9
  1057.6 1923.52  1077.7 1926.81  1128.1 1933.63  1178.5 1938.81    1239 1943.29
#Mann= 3 , 0 , 0
       0     .11       0   581.3    .045       0   596.3     .11       0
Bank Sta=581.3,596.3
XS Rating Curve= 0 ,0
Exp/Cntr=0.3,0.1

Type RM Length L Ch R = 1 ,14381.1 ,709.1,708.3,706.8
XS GIS Cut Line= 2
     2153157.827      270363.535     2154248.722      270215.295
#Sta/Elev= 30
       0 2082.12      20 2068.98      40  2055.3   100.1 2012.86   130.1 1992.11
   160.1 1972.27   200.2  1946.6   210.2 1939.53   250.2 1908.85   260.2 1901.93
   270.2  1895.8   280.2 1890.48   290.2    1886   300.2 1882.39   310.3 1879.77
   340.3 1873.46   350.3 1872.32   360.3 1872.28   384.2 1873.29   399.2 1873.91
   530.4  1880.3   640.5 1883.52   710.6  1884.8   750.6 1887.03   780.6 1889.72
   830.7  1896.3   880.7 1901.84  1050.9 1917.46  1070.9 1920.32  1100.9 1925.88
#Mann= 3 , 0 , 0
       0     .11       0   384.2    .045       0   399.2     .11       0
Bank Sta=384.2,399.2
XS Rating Curve= 0 ,0
Exp/Cntr=0.3,0.1

Type RM Length L Ch R = 1 ,13672.8 ,785.6,786.7,782.1
XS GIS Cut Line= 3
      2153317.47      270804.454     2153541.731      271002.108
      2154262.57      270858.112
#Sta/Elev= 30
       0 2012.35      10 2009.62    19.9 2006.44    39.9  1999.3    49.8 1995.22
    69.8 1985.61   109.6 1965.82   239.1 1906.35     269 1892.18     279 1888.09
     289 1885.38     309 1881.73   359.4 1874.42   377.1 1871.29   389.6 1869.57
   392.1  1869.5   399.6 1869.27   490.2 1872.78   520.5 1873.58   570.8 1874.11
   661.4 1874.09     742 1875.16   782.3 1876.15   792.3 1876.91   802.4 1878.17
   953.5 1900.58   963.5 1901.71   973.6 1902.26  1013.9 1903.08    1034 1904.99
#Mann= 3 , 0 , 0
       0     .11       0   377.1    .045       0   392.1     .11       0
Bank Sta=377.1,392.1
XS Rating Curve= 0 ,0
Exp/Cntr=0.3,0.1

Type RM Length L Ch R = 1 ,12886   ,672.5,678.7,687.9
XS GIS Cut Line= 2
     2153480.366      271672.283      2154374.28      271400.113
#Sta/Elev= 30
       0 2044.68    50.2 2011.71    70.3 1998.78   110.5 1973.79   170.8 1937.03
   180.9 1930.72     201 1917.06   241.1 1888.58   261.2 1875.31   271.3 1869.86
   281.3 1867.09   291.4 1866.63   321.5  1866.5   391.9 1867.13     412 1867.12
     432 1866.78   462.2 1865.74   472.2 1865.21   487.4  1863.9   502.4 1862.78
   512.4  1862.8   522.5 1863.34   542.6 1864.89   582.8  1867.5     633 1871.89
   663.1 1875.33   703.3 1880.48   783.7 1890.32     844 1896.12   934.4 1905.65
#Mann= 3 , 0 , 0
       0     .11       0   487.4    .045       0   502.4     .11       0
Bank Sta=487.4,502.4
XS Rating Curve= 0 ,0
Exp/Cntr=0.3,0.1

Type RM Length L Ch R = 1 ,12207.4 ,590.6,574.9,559.5
XS GIS Cut Line= 2
     2153786.767      272086.925     2154668.037      272029.001
#Sta/Elev= 30
       0 1914.08    50.2 1888.85    60.2 1885.07    80.3 1879.45   110.4  1872.1
   130.5 1868.02   140.5 1866.41   150.5 1865.29   160.6 1864.65   210.8 1862.54
     281 1860.04   311.1 1859.22   411.5 1854.36   428.7 1853.82   431.6 1853.78
   443.7 1853.99   481.7 1855.33   531.9 1857.63   592.1 1860.59   602.2 1861.41
   612.2 1862.74   622.2 1864.52   652.3 1870.63   682.4 1876.36   712.6 1880.96
   732.6 1883.41   762.7  1886.4   792.8 1888.58     823 1890.52   883.2  1893.7
#Mann= 3 , 0 , 0
       0     .12       0   428.7    .045       0   443.7     .12       0
Bank Sta=428.7,443.7
XS Rating Curve= 0 ,0
Exp/Cntr=0.3,0.1

Type RM Length L Ch R = 1 ,11632.5 ,986.1,995.1,1002.6
XS GIS Cut Line= 2
     2154085.277      272868.412     2154758.059      272226.038
#Sta/Elev= 30
       0 1987.65      10 1983.33      60  1960.9      80 1952.17     130 1930.64
     160 1918.08     180 1909.96     200 1902.09   260.1 1879.08   290.1 1867.36
   300.1 1864.42   310.1 1862.72   390.1 1854.46   413.2 1851.91   420.1 1851.21
   428.2 1850.96   430.1  1850.9   550.1 1851.85   590.1 1852.31   660.1 1853.64
   750.2 1855.77   760.2  1856.1   770.2 1857.01   780.2 1858.67   820.2 1866.61
   850.2 1873.07   860.2 1875.09   870.2 1876.52   880.2 1877.66   930.2 1882.64
#Mann= 3 , 0 , 0
       0     .12       0   413.2    .045       0   428.2     .12       0
Bank Sta=413.2,428.2
XS Rating Curve= 0 ,0
Exp/Cntr=0.3,0.1

Type RM Length L Ch R = 1 ,10637.4 ,635.7,636.3,636.9
XS GIS Cut Line= 2
     2154381.757      273419.561      2155240.79      273077.468
#Sta/Elev= 30
       0 1945.79    40.2 1922.57    60.3  1911.7    90.4 1896.44   120.6 1882.62
   150.8 1869.79   160.8  1865.9   170.9 1862.52   180.9 1859.74   211.1 1852.56
   221.1 1851.28   301.5 1846.11   321.6 1845.19   422.1 1843.68   613.1 1841.82
   642.8 1840.99   653.3  1840.6   657.8  1840.7   663.3 1840.82   693.5 1843.25
   753.8 1847.32   773.9 1850.31   824.1 1860.28   854.3 1863.83   864.3 1865.53
   874.4 1867.76   894.5 1873.38   904.5 1875.67   914.6 1876.01   924.6 1875.25
#Mann= 3 , 0 , 0
       0     .12       0   642.8    .045       0   657.8     .12       0
Bank Sta=642.8,657.8
XS Rating Curve= 0 ,0
Exp/Cntr=0.3,0.1

Type RM Length L Ch R = 1 ,10001.1 ,742.8,748.5,754.2
XS GIS Cut Line= 2
     2154602.217      273894.689     2155639.897      273465.173
#Sta/Elev= 30
       0  1937.1   120.3 1892.38   150.4 1880.49   180.5 1867.93   190.5  1864.2
   220.6  1854.2   230.6 1851.33   240.7 1849.14   250.7 1847.84   260.7 1847.15
   320.9 1844.26   501.4 1838.53   631.7 1835.24   749.3 1833.49     752 1833.44
   762.1 1834.13   764.3 1834.86   772.1 1837.43   782.1 1843.66   792.2 1849.26
   802.2 1853.86   822.2 1862.67   832.3 1866.02   922.5 1886.09   942.6 1891.35
   952.6 1894.58   962.6 1898.44   982.7 1907.71    1103 1965.62  1123.1 1974.82
#Mann= 3 , 0 , 0
       0     .12       0   749.3    .045       0   764.3     .12       0
Bank Sta=749.3,764.3
XS Rating Curve= 0 ,0
Exp/Cntr=0.3,0.1

Type RM Length L Ch R = 1 ,9252.6  ,692.6,700.4,708
XS GIS Cut Line= 4
     2154514.793      274772.726     2155005.126      274309.001
     2155719.719      274198.771     2155780.535      273811.067
#Sta/Elev= 30
       0 2045.64    50.4 2016.98    70.5 2006.64     282 1914.06   302.2 1906.93
   322.3 1901.15   392.8 1884.02     413 1881.09   443.2 1878.89   493.6 1871.27
   533.9  1861.5   624.5 1842.18   644.7 1841.88   674.9 1843.96   725.1 1844.94
   785.4 1841.04   855.6 1840.64  1136.8 1824.45  1137.5 1824.52  1146.9 1825.41
  1152.5 1827.34    1177 1838.28  1197.1 1845.39  1307.6 1877.37  1357.8 1893.42
  1367.8 1895.64  1397.9 1899.36    1408 1901.44  1498.6 1923.49  1790.4 1987.75
#Mann= 3 , 0 , 0
       0     .12       0  1137.5    .045       0  1152.5     .12       0
Bank Sta=1137.5,1152.5
XS Rating Curve= 0 ,0
Exp/Cntr=0.3,0.1

Type RM Length L Ch R = 1 ,8552.2  ,779.7,779.3,779.1
XS GIS Cut Line= 2
     2154682.039      274753.721     2155847.201      274970.705
#Sta/Elev= 30
       0 1984.06    50.2 1952.66   110.5 1916.39   120.5 1910.49   170.8 1882.64
   180.8 1876.91   200.9 1864.01   210.9    1859     221 1855.65     231 1853.59
   241.1  1852.1   281.2 1847.05   351.5 1840.14   381.7 1836.68   441.9 1828.07
     462 1824.48   477.3 1821.22   492.3 1818.26   502.2 1817.45   522.3 1817.94
   602.6    1822   803.5 1828.17   883.9 1828.64   893.9 1829.55     904 1831.94
     914 1835.61  1014.4 1875.09  1124.9 1916.04  1155.1 1928.04  1185.2 1940.68
#Mann= 3 , 0 , 0
       0      .1       0   477.3    .045       0   492.3      .1       0
Bank Sta=477.3,492.3
XS Rating Curve= 0 ,0
Exp/Cntr=0.3,0.1

Type RM Length L Ch R = 1 ,7772.9  ,1060.4,1059,1057.4
XS GIS Cut Line= 2
     2154549.003      275521.529     2155864.158       275749.59
#Sta/Elev= 30
       0 2001.25    20.1 1991.19    40.1 1982.83    60.2 1975.22    90.3 1965.25
   150.5 1947.19   170.6 1940.02   190.7 1931.35   210.8 1920.73   240.9 1902.32
   361.3 1823.68   371.3 1818.41   381.4 1815.27   393.3 1813.42   408.3 1812.38
   411.5 1812.28   441.6 1812.55   491.8 1816.58   592.1 1818.33   903.2 1819.24
   913.3  1819.4   933.3 1820.89   983.5 1828.88  1063.8 1842.71  1134.1 1855.63
  1174.2 1863.76  1214.4 1872.76  1264.5 1885.42  1304.7 1897.22  1334.8 1907.22
#Mann= 3 , 0 , 0
       0      .1       0   393.3    .045       0   408.3      .1       0
Bank Sta=393.3,408.3
XS Rating Curve= 0 ,0
Exp/Cntr=0.3,0.1

Type RM Length L Ch R = 1 ,6713.9  ,1356.1,1358.5,1360.5
XS GIS Cut Line= 2
     2154552.189      276555.336     2155681.709      276658.036
#Sta/Elev= 30
       0 1992.45    90.3 1953.51   110.4 1944.04   130.5 1933.67   140.5 1928.89
   160.6 1920.44   170.6 1916.89   180.7 1914.25   210.8 1908.64     271    1894
   301.1 1888.14   311.2 1885.78   331.2 1879.38   341.3 1875.34   351.3 1870.49
   361.3 1864.58   371.4 1857.89   381.4 1850.54   391.4 1839.44   401.5 1823.08
   411.5 1813.63   421.6 1812.28   430.2 1812.28   445.2 1812.28   782.9 1812.46
   973.6 1819.96  1023.8 1821.41  1053.9 1821.36    1074  1821.8  1134.2 1824.42
#Mann= 3 , 0 , 0
       0      .1       0   430.2    .045       0   445.2      .1       0
Bank Sta=430.2,445.2
XS Rating Curve= 0 ,0
Exp/Cntr=0.3,0.1

Type RM Length L Ch R = 1 ,5355.4  ,1165,1163.9,1163.8
XS GIS Cut Line= 2
      2154357.22      277735.303     2155742.525      277976.992
#Sta/Elev= 30
       0 1908.82    50.2 1879.67    70.3 1868.81   100.4 1854.08   120.5 1844.67
   160.7 1827.04   170.8 1823.29   180.8 1820.98   190.8 1820.07   200.9 1819.56
   271.2 1816.95   371.6 1812.57   391.7 1812.28   742.6 1812.28   757.6 1812.28
   944.2  1812.3   954.2 1812.56   964.3 1813.48   994.4 1818.36  1024.5 1822.51
  1235.5 1845.36  1265.6 1847.67  1275.6 1848.72  1285.7  1850.3  1295.7 1852.37
  1305.8 1855.09  1325.9 1861.19  1335.9  1863.9  1376.1 1873.64  1406.2 1881.28
#Mann= 3 , 0 , 0
       0      .1       0   742.6    .045       0   757.6      .1       0
Bank Sta=742.6,757.6
XS Rating Curve= 0 ,0
Exp/Cntr=0.3,0.1

Type RM Length L Ch R = 1 ,4191.5  ,1043.8,1047.9,1051
XS GIS Cut Line= 2
     2154099.474        278817.7      2155507.25       279057.24
#Sta/Elev= 30
       0  1838.5    20.1 1837.29    40.2 1836.44    60.3 1835.17   130.7 1828.68
   201.1    1823   271.5 1818.42   321.8 1815.73   372.1 1812.68   382.1 1812.36
   392.2 1812.29   622.9 1812.28   637.9 1812.28  1025.8 1812.27  1035.8 1812.35
  1045.9 1813.45  1055.9 1815.15  1086.1 1818.73  1116.3 1822.66  1216.8 1836.55
  1277.2 1844.64  1297.3 1847.59  1307.3 1849.51  1317.4 1852.07  1347.6  1861.5
  1357.6 1864.46  1377.7 1870.19  1387.8 1872.78  1407.9 1877.08    1428 1880.87
#Mann= 3 , 0 , 0
       0      .1       0   622.9    .045       0   637.9      .1       0
Bank Sta=622.9,637.9
XS Rating Curve= 0 ,0
Exp/Cntr=0.3,0.1

Type RM Length L Ch R = 1 ,3143.7  ,340.3,337.3,334.2
XS GIS Cut Line= 2
     2153606.348      279478.398     2155351.019      279942.123
#Sta/Elev= 30
       0 1861.88    80.7 1841.85     121 1831.58   161.4 1821.14   171.4 1818.74
   181.5 1816.99   211.8 1812.92   221.9 1812.34     232 1812.28  1154.3 1812.28
  1169.3 1812.28  1381.7 1812.28  1391.8 1812.58  1401.8 1813.87  1432.1 1821.19
  1472.4 1831.53  1482.5 1834.03  1502.7 1838.56  1512.8 1841.13  1522.9 1844.27
    1543    1851  1593.5 1866.76  1603.5  1870.1  1613.6 1873.83  1643.9 1886.23
  1674.1 1897.99  1694.3 1905.72  1704.4  1909.4  1764.9 1930.76  1805.2  1944.7
#Mann= 3 , 0 , 0
       0      .1       0  1154.3    .045       0  1169.3      .1       0
Bank Sta=1154.3,1169.3
XS Rating Curve= 0 ,0
Exp/Cntr=0.3,0.1

Type RM Length L Ch R = 1 ,2806.4  ,170.9,167.3,163.7
XS GIS Cut Line= 4
     2152834.594      279630.125     2153511.508      279960.587
     2155137.166      280157.798      2155467.87      280030.644
#Sta/Elev= 30
       0 1977.96   130.6 1974.26   321.4 1961.21   331.4 1958.55   381.7  1939.8
   441.9 1915.61   512.2 1886.21   532.3 1878.76   753.3 1821.81   783.4 1815.63
   803.5 1812.66  1873.8 1812.28 1880.75 1811.46  1888.8 1812.28  2179.9 1812.33
    2200 1814.26  2240.2 1821.65  2300.4  1825.6  2310.5 1828.16  2320.5 1832.47
  2350.7 1848.67  2360.7 1852.97  2390.8 1862.42  2459.7 1898.17  2479.4 1906.93
  2499.1 1914.71  2528.6 1925.25  2558.2 1934.26  2666.4 1963.81  2745.2 1989.86
#Mann= 3 , 0 , 0
       0      .1       0  1873.8    .045       0  1888.8      .1       0
#XS Ineff= 2 , 0
         1800.54 1815.78 1949.87         1816.82
Permanent Ineff=
       F       F
Bank Sta=1873.8,1888.8
XS Rating Curve= 0 ,0
Exp/Cntr=0.3,0.1

Type RM Length L Ch R = 1 ,2639.1  ,614.3,617.6,620.9
XS GIS Cut Line= 5
     2153213.026      280331.024     2153588.793      280283.054
     2154777.389      280253.739     2155329.047      280277.724
     2155462.298      280144.473
#Sta/Elev= 30
       0 1830.91    69.8 1827.89   139.6 1822.15   239.2 1824.16   289.1 1821.87
   388.9 1809.42   419.1 1804.04   469.5 1792.22   509.8 1784.46   560.2 1778.01
   590.4 1775.62   812.1 1774.17   963.2 1776.08  1245.4  1775.6  1315.9 1777.54
  1346.1 1776.23  1376.3 1771.82  1396.5 1769.84  1416.6 1772.24  1477.1 1795.94
  1497.2 1800.84  1768.6 1829.73  1838.8 1833.97  1939.2 1837.08  2029.6 1844.92
    2120 1855.22  2179.5 1889.61    2239 1926.99  2258.8 1936.85  2308.4 1958.49
#Mann= 3 , 0 , 0
       0      .1       0  1376.3    .045       0  1416.6      .1       0
#XS Ineff= 2 , 0
          1203.4 1799.45
Permanent Ineff=
       F       F
Bank Sta=1376.3,1416.6
XS Rating Curve= 0 ,0
Exp/Cntr=0.3,0.1

Type RM Length L Ch R = 1 ,2021.5  ,263.2,249.4,248.3
XS GIS Cut Line= 4
     2152796.096      280135.342       2153921.2       280784.05
     2154868.922      280885.411     2155639.264      280059.321
#Sta/Elev= 30
       0 1999.95    50.3  1985.5   120.8 1960.27   171.2 1939.22     302 1877.85
   362.4 1854.12   402.7 1840.99   483.2 1827.12   563.8 1823.95   654.4  1813.3
   724.9 1797.02   805.4 1796.87   855.8 1779.84   875.9 1776.92  1730.1  1776.3
  1750.2 1774.17  1769.8 1767.04  1784.8 1766.82  1820.4 1772.94  1950.9 1773.62
  2161.6 1765.35  2483.8 1765.21  2836.8 1777.48    2857 1780.78  2957.8 1839.08
    2978 1843.36  3018.3 1838.72  3038.5 1844.59  3179.7 1935.24  3381.4 2026.39
#Mann= 3 , 0 , 0
       0      .1       0  1769.8    .045       0  1784.8      .1       0
#XS Ineff= 2 , 0
                         1931.98         1784.64
Permanent Ineff=
       F       F
Bank Sta=1769.8,1784.8
XS Rating Curve= 0 ,0
Exp/Cntr=0.3,0.1

Type RM Length L Ch R = 1 ,1772.1  ,1753.9,1772.1,1777.6
XS GIS Cut Line= 4
     2152737.144      280331.412     2154096.469      281057.976
     2155130.652      281143.247     2155985.548      280124.369
#Sta/Elev= 30
       0  1917.7   151.1 1897.98   201.5 1883.14   302.2  1846.5     403 1824.38
   453.3 1822.76   493.6 1814.72   614.5  1798.5     675 1796.02   735.4 1777.87
  1470.8  1776.5  1541.3 1772.18  1692.4 1770.12  1783.1 1763.45  1785.1  1763.5
  1800.1 1763.96  1954.4 1766.55  2014.8  1771.7  2125.6 1766.61    2579 1770.87
  3042.5 1768.33  3274.2 1781.67  3415.3 1792.94  3445.5 1798.06  3475.8 1808.85
  3536.2 1837.06  3657.1 1862.88  3757.9 1879.65  3858.6 1910.93    3909 1921.68
#Mann= 3 , 0 , 0
       0      .1       0  1785.1    .045       0  1800.1      .1       0
Bank Sta=1785.1,1800.1
XS Rating Curve= 0 ,0
Exp/Cntr=0.3,0.1

Chan Stop Cuts=-1
Use User Specified Reach Order=0
